--- P155-00-00.PRJ (project) ---

Proj Title=P155-00-00
Current Plan=p02
Default Exp/Contr=.3,.1
English Units
Geom File=g01
Flow File=f02
Flow File=f01
Plan File=p04
Plan File=p03
Plan File=p02
Plan File=p01
Y Axis Title=Elevation
X Axis Title(PF)=Main Channel Distance
X Axis Title(XS)=Station
BEGIN DESCRIPTION:
Greens Bayou Watershed
P155-00-00
HCFCD Unit P155-00-00
Flood Hazard Model
10, 2, 1, 0.2% Event
Filename P155-00-00.prj
Prepared by:  Watershed Concepts  Date:
Reviewed by:                      Date:
STATUS FINAL
END DESCRIPTION:
DSS Export Rating Curves= 0
DSS Export Rating Curve Sorted= 0
DSS Export Volume Flow Curves= 0
DXF OffsetX= 0
DXF OffsetY= 0
DXF ScaleX= 1
DXF ScaleY= 10

--- P155-00-00.p02 (plan) ---

Plan Title=Floodway
Version=Version 3.0.1  Mar 2001
Short Identifier=Floodway060
Geom File=g01
Flow File=f02
Subcritical Flow
K Sum by GR= 0
Std Step Tol= 0.01
Critical Tol= 0.01
Num of Std Step Trials= 20
Max Error Tol= 0.3
Flow Tol Ratio= 0.001
Split Flow NTrial= 30
Split Flow Tol= 0.02
Split Flow Ratio= 0.02
Log Output Level= 0
Friction Slope Method= 1
Unsteady Friction Slope Method= 2
Parabolic Critical Depth
Global Vel Dist= 0 , 0 , 0
Global Log Level= 0
CheckData=True
Encroach Param=-1 ,0,0, 2
Encroach River=P155-00-00
Encroach Reach=Reach - 1
Encroach Node=7191.1
       1  4945.4  5049.9
Encroach Node=6618.3
       1  4947.3  5053.7
Encroach Node=6298.5
       1  4947.3  5053.7
Encroach Node=5602.1
       1  4945.7  5050.2
Encroach Node=5465.6
       1  4945.7  5050.2
Encroach Node=4618.7
       1  4941.6  5047.4
Encroach Node=4013.9
       1  4948.5  5049.5
Encroach Node=3917.0
       1  4948.5  5049.5
Encroach Node=3866.0
       1  4948.5  5049.5
Encroach Node=3815.0
       1  4948.5  5049.5
Encroach Node=3604.3
       1  4949.9  5049.4
Encroach Node=3583.9
       1  4949.9  5049.4
Encroach Node=3565.8
       1  4950.9  5050.3
Encroach Node=3147.1
       1 4948.35 5051.65
Encroach Node=2443.1
       1 4948.35 5051.65
Encroach Node=1720.0
       1    4963    5060
Encroach Node=1467.7
       1    4956    5049
Encroach Node=1390.9
       1    4970    5030
Encroach Node=1324.6
       1    4970    5030
Encroach Node=1258.3
       1    4970    5030
Encroach Node=1141.6
       1    4950    5050
Encroach Node=1124.5
       1    4950    5050
Encroach Node=1107.4
       1    4950    5050
Encroach Node=898.1
       1    4925    5050
Encroach Node=840.2
       1    4966    5028
Encroach Node=812.0
       1    4966    5028
Encroach Node=783.8
       1    4966    5028
Encroach Node=513.6
       1  4975.1    5025
Encroach Reach=P155-00-00_0005
Encroach Node=7191.1
       1  4945.4  5049.9
Encroach Node=6618.3
       1  4947.3  5053.7
Encroach Node=6298.5
       1  4947.3  5053.7
Encroach Node=5602.1
       1  4945.7  5050.2
Encroach Node=5465.6
       1  4945.7  5050.2
Encroach Node=4618.7
       1  4941.6  5047.4
Encroach Node=4013.9
       1  4948.5  5049.5
Encroach Node=3917.0
       1  4948.5  5049.5
Encroach Node=3866.0
       1  4948.5  5049.5
Encroach Node=3815.0
       1  4948.5  5049.5
Encroach Node=3604.3
       1  4949.9  5049.4
Encroach Node=3583.9
       1  4949.9  5049.4
Encroach Node=3565.8
       1  4950.9  5050.3
Encroach Node=3147.1
       1 4948.35 5051.65
Encroach Node=2443.1
       1 4948.35 5051.65
Encroach Node=1720.0
       1    4963    5060
Encroach Node=1467.7
       1    4956    5049
Encroach Node=1390.9
       1    4970    5030
Encroach Node=1324.6
       1    4970    5030
Encroach Node=1258.3
       1    4970    5030
Encroach Node=1141.6
       1    4950    5050
Encroach Node=1124.5
       1    4950    5050
Encroach Node=1107.4
       1    4950    5050
Encroach Node=898.1
       1    4925    5050
Encroach Node=840.2
       1    4966    5028
Encroach Node=812.0
       1    4966    5028
Encroach Node=783.8
       1    4966    5028
Encroach Node=513.6
       1  4975.1    5025
Computation Interval=1HOUR
Output Interval=1HOUR
Run HTab= 0
Run UNet= 0
Run PostProcess= 0
UNET Theta= 1
UNET ZTol= 0.02
UNET ZSATol= 0.1
UNET MxIter= 20
UNET MaxInSteps= 20
UNET DtIC= 0
UNET DtMin= 0
UNET MaxCRTS= 20
UNET WFStab= 2
UNET SFStab= 1
UNET WFX= 1
UNET SFX= 1
UNET Convert EG Bridges=-1
UNET Use Existing IB Tables=-1
Instantaneous Interval=1HOUR
Write IC File= 0
IC Time=0
Write Velocity= 0
Write Detailed= 0

--- P155-00-00.p01 (plan) ---

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Plan Title=FEMA Effective June 2007
Short Identifier=FEMAeff0607
Geom File= g01
Flow File= f01
Interactive Comp Mode
Encroach Param= -1, 0, 0, 0

--- P155-00-00.p03 (plan) ---

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Plan Title=Floodway-Revised 081709
Short Identifier=Fldway-K WS
Geom File=g01
Flow File=f03
BEGIN DESCRIPTION:
Revised BC to Known WS (PBS&J Aug 09)
END DESCRIPTION:

--- P155-00-00.p04 (plan) ---

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Plan Title=FEMA Effective - Revised 081709
Short Identifier=FEMAeffBCkWS
Geom File=g01
Flow File=f01
Encroach Param=-1 ,0,0, 0
BEGIN DESCRIPTION:
Revised BC to Known WS (PBS&J - Aug 09)
END DESCRIPTION:

--- P155-00-00.f02 (steady flow) ---

Flow Title= Floodway
Number of Profiles= 2
Profile Names=1PCT_100yr, 1PCTFloodway_100yrFW
River Rch & RM=P155-00-00,P155-00-00_0005,7191.1
    1213    1213
River Rch & RM=P155-00-00,P155-00-00_0005,6618.3
    1261    1261
River Rch & RM=P155-00-00,P155-00-00_0005,6298.5
    1370    1370
River Rch & RM=P155-00-00,P155-00-00_0005,5602.1
    1393    1393
River Rch & RM=P155-00-00,P155-00-00_0005,5465.6
    1542    1542
River Rch & RM=P155-00-00,P155-00-00_0005,4618.7
    1658    1658
River Rch & RM=P155-00-00,P155-00-00_0005,4013.9
    1677    1677
River Rch & RM=P155-00-00,P155-00-00_0005,3917
    2357    2357
River Rch & RM=P155-00-00,P155-00-00_0005,3147.1
    2503    2503
River Rch & RM=P155-00-00,P155-00-00_0005,2443.1
    2604    2604
River Rch & RM=P155-00-00,P155-00-00_0005,1720
    2651    2651
River Rch & RM=P155-00-00,P155-00-00_0005,1390.9
    2692    2692
River Rch & RM=P155-00-00,P155-00-00_0005,1141.6
    2740    2740
River Rch & RM=P155-00-00,P155-00-00_0005,840.2
    2781    2781
Boundary for River Rch & Prof#=P155-00-00,P155-00-00_0005, 1
Up Type= 0
Dn Type= 3
Dn Slope= 0.00130
Boundary for River Rch & Prof#=P155-00-00,P155-00-00_0005, 2
Up Type= 0
Dn Type= 1
Dn Known WS=73.39

--- P155-00-00.f01 (steady flow) ---

Flow Title= FEMA Effective June 2007
Number of Profiles= 4
Profile Names=10PCT_10yr, 2PCT_50yr, 1PCT_100yr, 0.2PCT_500yr
River Rch & RM=P155-00-00,P155-00-00_0005,7191.1
     744    1062    1213    1714
River Rch & RM=P155-00-00,P155-00-00_0005,6618.3
     773    1103    1261    1779
River Rch & RM=P155-00-00,P155-00-00_0005,6298.5
     840    1199    1370    1928
River Rch & RM=P155-00-00,P155-00-00_0005,5602.1
     854    1218    1393    1959
River Rch & RM=P155-00-00,P155-00-00_0005,5465.6
     945    1347    1542    2161
River Rch & RM=P155-00-00,P155-00-00_0005,4618.7
    1016    1448    1658    2318
River Rch & RM=P155-00-00,P155-00-00_0005,4013.9
    1028    1465    1677    2344
River Rch & RM=P155-00-00,P155-00-00_0005,3917
    1439    2054    2357    3265
River Rch & RM=P155-00-00,P155-00-00_0005,3147.1
    1505    2177    2503    3452
River Rch & RM=P155-00-00,P155-00-00_0005,2443.1
    1549    2261    2604    3579
River Rch & RM=P155-00-00,P155-00-00_0005,1720
    1570    2301    2651    3639
River Rch & RM=P155-00-00,P155-00-00_0005,1390.9
    1588    2335    2692    3691
River Rch & RM=P155-00-00,P155-00-00_0005,1141.6
    1609    2376    2740    3751
River Rch & RM=P155-00-00,P155-00-00_0005,840.2
    1627    2410    2781    3802
Boundary for River Rch & Prof#=P155-00-00,P155-00-00_0005, 1
Up Type= 0
Dn Type= 3
Dn Slope= 0.00130
Boundary for River Rch & Prof#=P155-00-00,P155-00-00_0005, 2
Up Type= 0
Dn Type= 3
Dn Slope= 0.00130
Boundary for River Rch & Prof#=P155-00-00,P155-00-00_0005, 3
Up Type= 0
Dn Type= 3
Dn Slope= 0.00130
Boundary for River Rch & Prof#=P155-00-00,P155-00-00_0005, 4
Up Type= 0
Dn Type= 3
Dn Slope= 0.00130

--- P155-00-00.g01 (geometry) ---

Geom Title=P155-00-00 June 2007
Version=Version 3.0.1  Mar 2001

River Reach=P155-00-00      ,P155-00-00_0005
Reach XY= 30
      3117359.08     13916311.08      3117371.87     13916151.49
      3117371.75       13915904.      3117404.25       13915462.
        3117421.       13915417.      3117463.75       13915387.
       3117520.5       13915381.        3118039.       13915409.
      3118075.75       13915395.        3118114.       13915358.
      3118129.25       13915317.      3118140.52      13915234.2
       3118180.8      13914240.7      3118237.99     13913265.58
      3118269.75       13912439.      3118260.75       13912371.
      3118242.25       13912318.        3118210.       13912267.
        3118155.       13912207.      3118096.75       13912158.
      3118020.75       13912125.        3117883.       13912114.
      3117751.25       13912114.      3117559.75       13912097.
       3117458.5       13912054.      3117375.75       13911982.
        3117319.       13911909.      3117119.75       13911527.
      3117115.25       13911487.      3117140.75       13911002.

Type RM Length L Ch R = 1 ,7191.1  ,575.1,572.8,568.5
BEGIN DESCRIPTION:
Cross Section 7191.1
END DESCRIPTION:
XS GIS Cut Line= 3
      3117459.09     13916323.11      3117361.31     13916311.26
      3117267.47     13916303.36
#Sta/Elev= 14
  4899.3    83.6  4919.3    82.8  4927.2   82.91  4945.4   83.13  4967.7   75.78
    4989   71.44  4991.5   70.94  5001.7   70.68  5010.2   71.04  5010.9   71.44
  5049.9   83.65  5083.6   83.47  5087.8    84.3    5092    84.4
#Mann= 5 , 1 , 0
  4899.3      .2       0  4899.3      .1       0  4945.4    .035       0
  5049.9     .14       0    5092      .2       0
Bank Sta=4945.4,5049.9
XS Rating Curve= 0
Exp/Cntr=.3,.1

Type RM Length L Ch R = 1 ,6618.3  ,306.9,319.8,337.2
BEGIN DESCRIPTION:
Cross Section 6618.3
END DESCRIPTION:
XS GIS Cut Line= 2
      3117503.82     13915746.93      3117264.11      13915731.6
#Sta/Elev= 16
  4879.8    83.3  4909.8    82.6  4939.8    83.1  4947.3   81.07  4949.8    80.4
  4977.6    73.4    4989   71.24  4990.3   70.05  5009.2   70.22  5011.1   71.29
  5019.2   72.93    5031   74.88  5039.8    81.8  5049.8    83.7  5053.7   83.68
    5120    83.3
#Mann= 3 , 1 , 0
  4879.8      .1       0  4947.3    .035       0  5053.7     .14       0
Bank Sta=4947.3,5053.7
XS Rating Curve= 0
Exp/Cntr=.3,.1

Type RM Length L Ch R = 1 ,6298.5  ,682.5,696.4,660.9
BEGIN DESCRIPTION:
Cross Section 6298.5-Interpolated
END DESCRIPTION:
XS GIS Cut Line= 4
      3117746.32     13915597.33      3117487.22       13915455.
      3117363.12      13915396.6      3117308.32     13915374.68
#Sta/Elev= 20
  4628.8    83.4  4718.8    82.8  4768.8    81.9  4878.8    83.2  4908.8    82.2
  4924.5    82.5  4930.1   82.33  4947.3   82.61  4977.6   73.15    4989   70.99
  4990.3    69.8  5009.2   69.97  5011.1   71.04  5019.2   72.68    5031   74.63
  5053.7   82.32  5067.3    82.3  5071.6    82.1  5091.6    83.2  5120.6    83.8
#Mann= 5 , 1 , 0
  4628.8      .2       0  4628.8      .1       0  4947.3    .017       0
  5053.7     .14       0  5120.6      .2       0
Bank Sta=4947.3,5053.7
XS Rating Curve= 0
Exp/Cntr=.3,.1

Type RM Length L Ch R = 1 ,5602.1  ,168.9,136.5,110.5
BEGIN DESCRIPTION:
Cross Section 5602.1-Interpolated
END DESCRIPTION:
XS GIS Cut Line= 4
      3118333.98     13915560.83      3118140.55      13915418.5
      3118049.31      13915345.5      3117828.82     13915280.04
#Sta/Elev= 23
  4697.4    82.4  4737.4    82.3  4757.4    81.5  4807.4    82.1  4827.4    81.6
  4867.4      82  4875.4   81.68  4877.4    81.6  4917.4    82.3  4937.6    81.8
  4945.7    81.4    4967    73.9  4995.6   69.32  4996.2   68.68  4999.4   68.28
  5002.3      68  5004.4   68.36  5027.4   73.86  5050.2   81.54  5054.4    81.7
  5064.4    82.5  5124.4    80.9  5284.4    83.6
#Mann= 5 , 1 , 0
  4697.4      .2       0  4697.4      .1       0  4875.4     .05       0
  4945.7    .017       0  5050.2     .05       0
Bank Sta=4945.7,5050.2
XS Rating Curve= 0
Exp/Cntr=.3,.1

Type RM Length L Ch R = 1 ,5465.6  ,843.9,846.9,851.8
BEGIN DESCRIPTION:
Cross Section 5465.6
END DESCRIPTION:
XS GIS Cut Line= 4
      3118401.12     13915262.68      3118372.99     13915258.18
      3117797.21     13915252.18      3117547.29     13915245.93
#Sta/Elev= 22
  4736.1      81  4764.6    80.7  4819.5   80.82  4854.6    80.9  4909.5   81.23
  4925.1   79.57  4945.7   81.21    4967   73.71  4995.6   69.13  4996.2   68.49
  4999.4   68.09  5002.3   67.81  5004.4   68.17  5027.4   73.67  5050.2   81.35
  5063.9    81.6  5084.8   81.83  5094.6    82.6  5164.6    81.9  5294.6    82.3
  5488.5    82.5  5590.4    82.6
#Mann= 5 , 1 , 0
  4736.1     .14       0  4819.5     .07       0  4945.7    .035       0
  5050.2     .07       0  5488.5      .1       0
#XS Ineff= 2 , 0
       0  4945.7   81.21               0
Permanent Ineff=
       F       F
Bank Sta=4945.7,5050.2
XS Rating Curve= 0
Exp/Cntr=.3,.1

Type RM Length L Ch R = 1 ,4618.7  ,609.1,604.8,602.7
BEGIN DESCRIPTION:
Cross Section 4618.7
END DESCRIPTION:
XS GIS Cut Line= 3
      3118389.44     13914419.18      3118103.09     13914406.52
      3117584.09     13914373.09
#Sta/Elev= 23
  4784.3    81.6  4794.3    81.7  4814.3    81.3  4864.3    81.6  4904.3    81.3
  4908.4   81.34  4922.6   80.56  4941.6   81.24  4957.7    75.1    4995   68.86
  4996.6   67.57  4999.5   67.51  5003.7   68.13  5004.9    68.9  5006.4   69.45
  5047.4   81.72  5059.6   81.58  5073.6   80.94    5101    80.3    5221    80.7
    5361    80.8    5561    80.5    5591    81.6
#Mann= 3 , 1 , 0
  4784.3     .14       0  4941.6    .035       0  5047.4      .1       0
Bank Sta=4941.6,5047.4
XS Rating Curve= 0
Exp/Cntr=.3,.1

Type RM Length L Ch R = 1 ,4013.9  ,100.8,96.9,95.7
BEGIN DESCRIPTION:
Cross Section 4013.9-Interpolated
END DESCRIPTION:
XS GIS Cut Line= 4
      3118309.31     13913803.61      3118265.86     13913803.61
      3118180.34     13913806.36      3117780.41     13913800.15
#Sta/Elev= 25
  4894.4    80.3  4934.4    79.1  4937.8    79.2  4947.8    79.5  4948.5   79.36
  4957.8    77.5  4967.8    74.5  4987.8    70.8  4997.8    69.4  4998.6   67.04
  5002.8   67.29  5004.1   67.97  5007.8    69.1  5017.8      70  5023.4    70.8
  5049.5    78.2  5053.4    79.3  5063.4    80.1  5083.4    80.8  5103.4    82.8
  5163.4    84.4  5343.4    84.2  5383.4    85.7  5403.4    85.6  5423.4    86.1
#Mann= 3 , 1 , 0
  4894.4     .14       0  4948.5    .035       0  5049.5      .1       0
Bank Sta=4948.5,5049.5
XS Rating Curve= 0
Exp/Cntr=.5,.3

Type RM Length L Ch R = 1 ,3917.0  ,102,102,102
BEGIN DESCRIPTION:
Upstream Section of Bridge/Culvert/Weir
END DESCRIPTION:
XS GIS Cut Line= 6
      3118832.42     13913628.75      3118663.21     13913633.47
       3118286.9     13913675.61      3118176.34     13913678.96
      3117925.06     13913695.71      3117740.93     13913690.59
#Sta/Elev= 22
  4376.2   79.62  4436.2   79.12  4474.5   78.37  4524.5   78.65  4664.5   77.22
  4752.4    75.8    4806   74.68  4869.6    79.1  4912.8   77.96  4948.5   78.69
  4984.1   70.16  4995.8    67.7  4998.6   66.97  5002.8   67.22  5004.1    67.9
    5011   68.87  5049.5   80.08    5129   80.71  5180.8   79.94  5332.2   79.31
  5430.8    80.9  5470.8   83.68
#Mann= 3 , 1 , 0
  4376.2     .14       0  4948.5     .03       0  5049.5      .1       0
#XS Ineff= 2 , 0
       0    4928    81.3    5060       0    86.4
Permanent Ineff=
       F       F
Bank Sta=4948.5,5049.5
XS Rating Curve= 0
Exp/Cntr=.5,.3

Type RM Length L Ch R = 3 ,3866.0  ,,,
BEGIN DESCRIPTION:
HARDY AIRPORT CONNECTOR
Structure ID: P55-5
END DESCRIPTION:
Bridge Culvert--1,0,-1,-1, 0
Deck Dist Width WeirC Skew NumUp NumDn MinLoCord MaxHiCord MaxSubmerge Is_Ogee
10,82,2.6,0, 55, 55, , , .95, 0, 1,1,,
  4376.2  4379.4  4436.2  4474.5  4499.4  4524.5  4664.5  4669.4  4679.4 4747.09
  4747.2 4747.31  4752.4    4806  4834.5  4869.6    4890  4912.8  4938.8 4938.91
    4939  4948.5  4984.1  4984.2  4993.2  4995.8    4997  4998.6  5002.8  5004.1
  5010.9    5011  5049.5 5050.09  5050.2  5050.4    5072  5074.2    5129  5149.7
  5180.8  5221.3  5268.6 5268.99  5269.1 5269.21  5269.5  5286.6  5332.2  5356.6
  5366.6  5420.8  5430.8  5466.6  5470.8
   79.61    81.1   81.15   81.18    81.2   81.24   81.49    81.5    81.8   82.59
   85.19   85.19   85.26   86.03   86.44   87.04   87.39   87.84   88.35   88.35
   88.35   88.52   89.12   89.13   89.28   89.33   89.35   89.38   89.46   89.49
   89.62   89.62   90.36   90.37   90.37   90.37   90.66   90.69   91.73   92.12
   92.95   94.03   95.65   95.66   95.66   93.06   93.07    86.3   87.34    87.9
    88.5   90.23   90.55    91.7   83.67
   79.61   79.58   79.11   78.36    78.5   78.64   77.21   77.13   76.97   75.88
   75.87   75.87   75.79   74.67   76.65   79.09   78.55   77.95   78.48   78.48
   80.42   80.59   81.19    81.2   81.35    81.4   81.42   81.45   81.53   81.56
   81.69   81.69   82.43   82.44   80.07   80.08   80.21   80.23    80.7   80.39
   79.93   79.76   79.57   79.57   79.57   79.57   79.57   79.49    79.3   79.69
   79.85   80.71   80.89   83.38   83.67
  4376.2  4379.4  4436.2  4474.5  4499.4  4524.5  4664.5  4669.4  4679.4 4747.09
  4747.2 4747.31  4752.4    4806  4834.5  4869.6    4890  4912.8  4938.8 4938.91
    4939  4948.5  4984.1  4984.2  4993.2  4995.8    4997  4998.6  5002.8  5004.1
  5010.9    5011  5049.5 5050.09  5050.2  5050.4    5072  5074.2    5129  5149.7
  5180.8  5221.3  5268.6 5268.99  5269.1 5269.21  5269.5  5286.6  5332.2  5356.6
  5366.6  5420.8  5430.8  5466.6  5470.8
   79.61    81.1   81.15   81.18    81.2   81.24   81.49    81.5    81.8   82.59
   85.19   85.19   85.26   86.03   86.44   87.04   87.39   87.84   88.35   88.35
   88.35   88.52   89.12   89.13   89.28   89.33   89.35   89.38   89.46   89.49
   89.62   89.62   90.36   90.37   90.37   90.37   90.66   90.69   91.73   92.12
   92.95   94.03   95.65   95.66   95.66   93.06   93.07    86.3   87.34    87.9
    88.5   90.23   90.55    91.7   83.67
   79.45   79.42   78.95    78.2   78.34   78.48   77.05   76.97   76.81   75.72
   75.71   75.71   75.63   74.51   76.49   78.93   78.39   77.79   78.32   78.32
   80.26   80.43   81.03   81.04   81.19   81.24   81.26   81.29   81.37    81.4
   81.53   81.53   82.27   82.28   79.91   79.92   80.05   80.07   80.54   80.23
   79.77    79.6   79.41   79.41   79.41   79.41   79.41   79.33   79.14   79.53
   79.69   80.55   80.73   83.22   83.51
Abutment Skew #Up #Dn= , 2 , 2
  4938.8  4984.2
   80.42   70.13
  4938.8  4984.2
   80.26   69.97
Abutment Skew #Up #Dn= , 2 , 2
    5011 5050.29
   68.86   82.44
    5011 5050.29
    68.7   82.28
BR Coef= 1 , 1 , 0 ,1.25, 0 ,,,.8,0,2,0,
WSPro=,,,, 1 ,,,, 0 ,,,, 0 ,,,,-1 ,-1 ,-1 , 0 , 0 , 0 , 0 , 0
BR U #Sta/Elev= 55
  4376.2   79.61  4379.4   79.58  4436.2   79.11  4474.5   78.36  4499.4    78.5
  4524.5   78.64  4664.5   77.21  4669.4   77.13  4679.4   76.97 4747.09   75.88
  4747.2   75.87 4747.31   75.87  4752.4   75.79    4806   74.67  4834.5   76.65
  4869.6   79.09    4890   78.55  4912.8   77.95  4938.8   78.48 4938.91   78.48
    4939   78.49  4948.5   78.68  4984.1   70.15  4984.2   70.13  4993.2   68.24
  4995.8   67.69    4997   67.37  4998.6   66.96  5002.8   67.21  5004.1   67.89
  5010.9   68.85    5011   68.86  5049.5   80.07 5050.09   80.07  5050.2   80.07
  5050.4   80.08    5072   80.21  5074.2   80.23    5129    80.7  5149.7   80.39
  5180.8   79.93  5221.3   79.76  5268.6   79.57 5268.99   79.57  5269.1   79.57
 5269.21   79.57  5269.5   79.57  5286.6   79.49  5332.2    79.3  5356.6   79.69
  5366.6   79.85  5420.8   80.71  5430.8   80.89  5466.6   83.38  5470.8   83.67
BR U #Mann= 3
  4376.2     .14  4948.5     .03  5049.5      .1
BR U Banks=4948.5,5049.5
BR D #Sta/Elev= 55
  4376.2   79.45  4379.4   79.42  4436.2   78.95  4474.5    78.2  4499.4   78.34
  4524.5   78.48  4664.5   77.05  4669.4   76.97  4679.4   76.81 4747.09   75.72
  4747.2   75.71 4747.31   75.71  4752.4   75.63    4806   74.51  4834.5   76.49
  4869.6   78.93    4890   78.39  4912.8   77.79  4938.8   78.32 4938.91   78.32
    4939   78.33  4948.5   78.52  4984.1   69.99  4984.2   69.97  4993.2   68.08
  4995.8   67.53    4997   67.21  4998.6    66.8  5002.8   67.05  5004.1   67.73
  5010.9   68.69    5011    68.7  5049.5   79.91 5050.09   79.91  5050.2   79.91
  5050.4   79.92    5072   80.05  5074.2   80.07    5129   80.54  5149.7   80.23
  5180.8   79.77  5221.3    79.6  5268.6   79.41 5268.99   79.41  5269.1   79.41
 5269.21   79.41  5269.5   79.41  5286.6   79.33  5332.2   79.14  5356.6   79.53
  5366.6   79.69  5420.8   80.55  5430.8   80.73  5466.6   83.22  5470.8   83.51
BR D #Mann= 3
  4376.2     .14  4948.5     .03  5049.5      .1
BR D Banks=4948.5,5049.5
BC Design=,, 0 ,, 0 ,,,,,,

Type RM Length L Ch R = 1 ,3815.0  ,210.7,210.7,210.7
BEGIN DESCRIPTION:
Downstream Section of Bridge/Culvert/Weir
END DESCRIPTION:
XS GIS Cut Line= 6
      3118838.27     13913526.92      3118669.07     13913531.63
      3118292.76     13913573.77       3118182.2     13913577.12
      3117930.92     13913593.87      3117746.78     13913588.76
#Sta/Elev= 22
  4376.2   79.42  4436.2   78.92  4474.5   78.17  4524.5   78.45  4664.5   77.02
  4752.4    75.6    4806   74.48  4869.6    78.9  4912.8   77.76  4948.5   78.49
  4984.1   69.96  4995.8    67.5  4998.6   66.77  5002.8   67.02  5004.1    67.7
    5011   68.67  5049.5   79.88    5129   80.51  5180.8   79.74  5332.2   79.11
  5430.8    80.7  5470.8   83.48
#Mann= 3 , 1 , 0
  4376.2     .14       0  4948.5     .03       0  5049.5      .1       0
#XS Ineff= 2 , 0
       0    4928    81.1    5060       0    86.2
Permanent Ineff=
       F       F
Bank Sta=4948.5,5049.5
XS Rating Curve= 0
Exp/Cntr=.5,.3

Type RM Length L Ch R = 1 ,3604.3  ,38.5,38.5,38.5
BEGIN DESCRIPTION:
Cross Section 3604.3, Upstream Section of Weir
END DESCRIPTION:
XS GIS Cut Line= 2
      3118570.22     13913381.13      3118041.53     13913353.61
#Sta/Elev= 25
  4660.7    79.4  4690.7    78.8  4710.7    77.9  4770.7    77.7  4789.1      78
  4823.8   77.74  4853.6    78.4  4873.1   78.08  4889.7   79.21  4894.3   79.52
    4941   79.42  4949.9    79.4  4986.6    67.8  4995.7   66.87  4997.5   66.29
  4998.3   66.07    5003   66.25  5004.2   66.79  5013.9   68.26  5049.4   79.72
  5063.6   79.91  5078.4   79.21  5099.1   79.47    5135   80.34  5190.1    81.9
#Mann= 4 , 1 , 0
  4660.7     .99       0  4889.7     .14       0  4949.9     .03       0
  5049.4      .1       0
#XS Ineff= 2 , 0
       0                  5063.6       0   79.91
Permanent Ineff=
       F       F
Bank Sta=4949.9,5049.4
XS Rating Curve= 0
Exp/Cntr=.7,.5

Type RM Length L Ch R = 5 ,3583.9  ,,,
BEGIN DESCRIPTION:
SHEET PILE WEIR
Structure ID:
END DESCRIPTION:
IW Pilot Flow=0
#Inline Weir SE= 22
  4660.7    79.4  4690.7    78.8  4710.7    77.9  4770.7    77.7  4789.1      78
  4823.1    77.8    4854   78.28  4871.7   77.94  4899.4   79.37  4928.5   77.21
  4943.6   79.38  4974.3   79.38  4974.9   73.15  5025.2   73.15  5025.6   79.48
  5048.7   79.48  5050.3   79.82  5060.9   80.29  5074.6   78.19  5098.3   79.19
  5137.9   79.61  5190.1    81.9
IW Dist,WD,Coef,Skew,MaxSub,Min_El,Is_Ogee,SpillHt,DesHd
10,1,3,0,.95,, 0 ,,,1,1,

Type RM Length L Ch R = 1 ,3565.8  ,418.7,418.7,418.7
BEGIN DESCRIPTION:
Cross Section 3565.8, Downstream Section of Weir
END DESCRIPTION:
XS GIS Cut Line= 2
      3118542.77     13913342.66      3118044.18     13913314.27
#Sta/Elev= 25
  4690.7    78.8  4710.7    77.9  4770.7    77.7  4789.1      78  4823.1    77.8
    4854   78.28  4871.7   77.94  4880.7    78.4  4899.4   79.37  4943.6   79.38
  4950.9   79.39  4984.5   68.17  4988.6   66.79  4991.1   65.83  4996.2   64.87
  5002.9   64.79  5008.2   65.68  5011.5   66.74  5015.2   68.16  5050.3   79.82
  5060.9   80.29  5074.6   78.19  5098.3   79.19  5137.9   79.61  5190.1    81.9
#Mann= 4 , 1 , 0
  4690.7     .99       0  4880.7     .14       0  4950.9     .03       0
  5050.3      .1       0
#XS Ineff= 2 , 0
       0                  5060.9       0   80.29
Permanent Ineff=
       F       F
Bank Sta=4950.9,5050.3
XS Rating Curve= 0
Exp/Cntr=.7,.5

Type RM Length L Ch R = 1 ,3147.1  ,737.7,704,667.8
BEGIN DESCRIPTION:
Cross Section 3147.1-Interpolated
END DESCRIPTION:
XS GIS Cut Line= 5
      3119223.17     13913022.96      3118602.83     13912943.17
       3118312.1      13912940.2       3118239.1      13912940.2
      3117939.22     13912930.73
#Sta/Elev= 30
    4024    78.7    4174   78.31    4184   78.58    4214   77.84    4244   78.36
    4264   77.74    4344    77.9    4474   77.48    4504    78.1    4644   77.28
  4669.4   77.85  4719.4   77.84  4729.4   78.24  4809.4   77.11  4849.4   77.62
  4879.4    77.4  4889.4   78.09  4899.4   78.32  4940.2   78.14 4948.35   76.59
 4972.35   67.92 4987.75   66.23 5001.35    65.2 5024.55   68.44 5051.65    77.4
  5053.2   77.07  5063.2   79.06  5083.2   78.73  5103.2   79.52  5313.2   79.61
#Mann= 4 , 1 , 0
    4024      .2       0    4024     .14       0 4948.35     .03       0
 5051.65      .1       0
#XS Ineff= 2 , 0
       0  4899.4    77.5               0
Permanent Ineff=
       F       F
Bank Sta=4948.35,5051.65
XS Rating Curve= 0
Exp/Cntr=.3,.1

Type RM Length L Ch R = 1 ,2443.1  ,736.8,723.1,696.1
BEGIN DESCRIPTION:
Cross Section 2443.1
END DESCRIPTION:
XS GIS Cut Line= 5
      3119308.45     13912171.18      3118754.58      13911992.2
      3118293.96     13912173.38      3118075.93     13912357.62
       3117765.7     13912697.27
#Sta/Elev= 30
  3797.7   78.95  3811.1    78.7  3847.7   77.24  3897.7   77.47  3927.7   76.46
  4127.7   76.42  4227.7   77.11  4287.7   76.35  4379.8   76.88  4519.8   75.72
  4689.8   76.46  4759.8   75.72  4863.3   76.98  4904.7   77.45 4911.45   76.27
 4948.35   77.28 4972.35   68.61 5001.35   65.89 5024.55   69.13 5051.65   78.09
  5220.2   76.65  5240.2   77.26  5280.2   76.78  5340.2   78.08  5410.2    77.7
  5430.2   76.66  5470.2   76.75  5500.2   78.15  5600.2   78.87  5620.2   79.67
#Mann= 5 , 1 , 0
  3797.7      .1       0  3811.1     .14       0  4863.3      .1       0
 4948.35     .03       0 5051.65      .1       0
#XS Ineff= 2 , 0
       0  4904.7    77.3  5104.7       0    77.3
Permanent Ineff=
       F       F
Bank Sta=4948.35,5051.65
XS Rating Curve= 0
Exp/Cntr=.3,.1

Type RM Length L Ch R = 1 ,1720.0  ,247.9,252.3,343.3
BEGIN DESCRIPTION:
Cross Section 1720.0-Interpolaed
END DESCRIPTION:
XS GIS Cut Line= 5
      3118118.59     13911605.66      3117605.44     13911865.26
      3117538.32     13912045.97      3117501.82     13912144.52
       3117301.5     13912715.29
#Sta/Elev= 30
  4193.5    78.4  4223.5   76.97  4343.5   76.56  4363.5    77.3  4463.5   77.42
  4503.5    75.5  4613.5   76.55  4643.5   75.85  4723.5   76.42  4778.6   75.91
  4828.6   77.76  4878.6   78.27  4915.9      77  4938.6   76.24  4958.6   77.45
  4974.4   74.96  4990.5   68.08  4990.7   65.82    4993   63.88  4998.7   63.85
  5021.3   66.56  5051.3   75.46  5066.4   78.05  5086.4   76.38  5106.4   76.92
  5136.4   76.23  5326.4   77.53  5446.4   76.63  5486.4   78.19  5671.3   78.44
#Mann= 6 , 1 , 0
  4193.5      .2       0  4193.5     .07       0  4915.9      .1       0
  4974.4     .03       0  5051.3      .1       0  5671.3      .2       0
#XS Ineff= 2 , 0
       0  4828.6      77  5066.4       0      77
Permanent Ineff=
       F       F
Bank Sta=4974.4,5051.3
XS Rating Curve= 0
Exp/Cntr=.3,.1

Type RM Length L Ch R = 1 ,1467.7  ,69.4,76.8,79
BEGIN DESCRIPTION:
Cross Section 1467.7-Interpolated
END DESCRIPTION:
XS GIS Cut Line= 4
       3117396.8     13911823.76      3117325.73     13911861.26
       3117264.3     13911901.51      3117044.01     13912013.77
#Sta/Elev= 23
  4891.7    78.2    4900   77.66  4911.7    76.9  4931.7    77.1  4951.7    76.9
  4961.7      76  4974.4   74.25  4990.5   67.37  4990.7   65.11    4993   63.17
  4998.7   63.14  5004.9   63.66  5009.2   64.79    5010   67.91  5028.5   75.27
  5045.5      76  5051.7   76.87  5055.5    77.4  5065.5    77.9  5085.5    77.1
  5215.5    77.4  5265.5    77.2  5292.8      78
#Mann= 6 , 1 , 0
  4891.7     .07       0    4900     .08       0  4974.4     .03       0
  5028.5     .08       0  5051.7      .1       0  5292.8      .2       0
#XS Ineff= 2 , 0
       0  4891.7    78.2               0
Permanent Ineff=
       F       F
Bank Sta=4974.4,5028.5
XS Rating Curve= 0
Exp/Cntr=.5,.3

Type RM Length L Ch R = 1 ,1390.9  ,132.6,132.6,132.6
BEGIN DESCRIPTION:
Upstream Section of Bridge/Culvert/Weir
END DESCRIPTION:
XS GIS Cut Line= 6
      3117676.22     13911612.18      3117444.18     13911738.74
      3117371.18     13911779.69      3117278.59     13911829.55
      3117189.57     13911872.28      3116930.99     13911980.66
#Sta/Elev= 30
  4546.5   78.53  4596.5   77.03  4616.5   76.23  4656.5   75.93  4717.3   77.33
  4737.3   76.93  4757.3   77.03  4767.3   76.63  4817.3   78.33  4851.8   78.43
  4881.8   77.13  4917.4   77.61  4962.3   76.93  4974.4   74.04  4990.4   67.16
  4990.7    64.9    4993   62.96  4998.7   62.93  5004.9   63.45  5009.2   64.58
    5010    67.7  5028.5   75.06  5059.1   77.75    5120   77.32  5168.5   77.26
    5239   77.52  5302.3   77.03  5338.8   77.63  5358.8   77.63  5378.8   78.03
#Mann= 3 , 1 , 0
  4546.5     .99       0  4974.4     .02       0  5028.5      .1       0
#XS Ineff= 2 , 0
       0    4968    78.4    5031       0    76.9
Permanent Ineff=
       F       F
Bank Sta=4974.4,5028.5
XS Rating Curve= 0
Exp/Cntr=.5,.3

Type RM Length L Ch R = 3 ,1324.6  ,,,
BEGIN DESCRIPTION:
GREENS ROAD
Structure ID: P55-3
END DESCRIPTION:
Bridge Culvert--1,0,-1,-1, 0
Deck Dist Width WeirC Skew NumUp NumDn MinLoCord MaxHiCord MaxSubmerge Is_Ogee
10,112.6,2.6,0, 57, 57, , , .95, 0, 1,1,,
  4546.5  4596.5  4616.5  4656.5  4717.3  4737.3  4757.3  4758.8  4767.3  4800.7
  4817.3  4851.8  4858.2  4881.8 4894.09  4894.2 4894.31  4917.4  4925.7  4928.5
  4962.3  4974.4 4978.61  4978.7  4978.8  4990.4  4990.5  4990.7    4993  4998.7
  5004.9  5009.2  5009.9    5010 5021.09  5021.2  5021.3  5028.5  5051.6  5059.1
  5079.3 5103.89    5104 5104.11  5109.1    5120  5168.5  5187.7  5211.8    5239
  5239.9  5260.4  5302.3  5308.8  5338.8  5358.8  5378.8
    78.5      77    76.2    75.9    77.3    76.9      77   76.95   76.61   77.75
   78.31   78.41   78.13   77.18   77.32   79.72   79.72   79.98   80.08   80.07
   79.99   79.96   79.95   79.95   79.95   79.95   79.95   79.95   79.95   79.95
   79.94   79.94   79.94   79.94   79.94   79.94   79.94   80.04   80.34   80.25
   79.99   79.68   79.68   77.41   77.38    77.3   77.24   77.28   77.33    77.5
   77.49    77.4      77    77.1    77.6    77.6      78
    78.5      77    76.2    75.9    77.3    76.9      77   76.94    76.6   77.74
    78.3    78.4   78.12    77.1   77.27   77.27   77.27   77.58   77.49   77.46
    76.9   74.01    72.2   75.25   75.25   75.25   75.25   75.25   75.25   75.25
   75.24   75.24   75.24   75.24   75.24   72.13   72.17   75.03   77.06   77.72
   77.58    77.4    77.4    77.4   77.37   77.29   77.23   77.27   77.32   77.49
   77.48   77.32      77    77.1    77.6    77.6      78
  4546.5  4596.5  4616.5  4656.5  4717.3  4737.3  4757.3  4758.8  4767.3  4800.7
  4817.3  4851.8  4858.2  4881.8 4894.09  4894.2 4894.31  4917.4  4925.7  4928.5
  4962.3  4974.4 4978.61  4978.7  4978.8  4990.4  4990.5  4990.7    4993  4998.7
  5004.9  5009.2  5009.9    5010 5021.09  5021.2  5021.3  5028.5  5051.6  5059.1
  5079.3 5103.89    5104 5104.11  5109.1    5120  5168.5  5187.7  5211.8    5239
  5239.9  5260.4  5302.3  5308.8  5338.8  5358.8  5378.8
    78.5      77    76.2    75.9    77.3    76.9      77   76.95   76.61   77.75
   78.31   78.41   78.13   77.18   77.32   79.72   79.72   79.98   80.08   80.07
   79.99   79.96   79.95   79.95   79.95   79.95   79.95   79.95   79.95   79.95
   79.94   79.94   79.94   79.94   79.94   79.94   79.94   80.04   80.34   80.25
   79.99   79.68   79.68   77.41   77.38    77.3   77.24   77.28   77.33    77.5
   77.49    77.4      77    77.1    77.6    77.6      78
    78.3    76.8      76    75.7    77.1    76.7    76.8   76.74    76.4   77.54
    78.1    78.2   77.92    76.9   77.07   77.07   77.07   77.38   77.29   77.26
    76.7   73.81      72   75.05   75.05   75.05   75.05   75.05   75.05   75.05
   75.04   75.04   75.04   75.04   75.04   71.93   71.97   74.83   76.86   77.52
   77.38    77.2    77.2    77.2   77.17   77.09   77.03   77.07   77.12   77.29
   77.28   77.12    76.8    76.9    77.4    77.4    77.8
Abutment Skew #Up #Dn= , 2 , 2
  4978.5  4990.5
   75.25   66.38
  4978.5  4990.5
   75.05   66.18
Abutment Skew #Up #Dn= , 2 , 2
    5010 5021.29
   67.67   75.24
    5010 5021.29
   67.47   75.04
BR Coef= 1 , 1 , 0 ,1.25, 0 ,,,.8,0,2,0,
WSPro=,,,, 1 ,,,, 0 ,,,, 0 ,,,,-1 ,-1 ,-1 , 0 , 0 , 0 , 0 , 0
BR U #Sta/Elev= 57
  4546.5    78.5  4596.5      77  4616.5    76.2  4656.5    75.9  4717.3    77.3
  4737.3    76.9  4757.3      77  4758.8   76.94  4767.3    76.6  4800.7   77.74
  4817.3    78.3  4851.8    78.4  4858.2   78.12  4881.8    77.1 4894.09   77.27
  4894.2   77.27 4894.31   77.27  4917.4   77.58  4925.7   77.49  4928.5   77.46
  4962.3    76.9  4974.4   74.01 4978.61    72.2  4978.7   72.16  4978.8   72.12
  4990.4   67.13  4990.5   66.38  4990.7   64.87    4993   62.93  4998.7    62.9
  5004.9   63.42  5009.2   64.55  5009.9   67.28    5010   67.67 5021.09   72.08
  5021.2   72.13  5021.3   72.17  5028.5   75.03  5051.6   77.06  5059.1   77.72
  5079.3   77.58 5103.89    77.4    5104    77.4 5104.11    77.4  5109.1   77.37
    5120   77.29  5168.5   77.23  5187.7   77.27  5211.8   77.32    5239   77.49
  5239.9   77.48  5260.4   77.32  5302.3      77  5308.8    77.1  5338.8    77.6
  5358.8    77.6  5378.8      78
BR U #Mann= 3
  4546.5     .99  4974.4     .02  5028.5      .1
BR U Banks=4974.4,5028.5
BR D #Sta/Elev= 57
  4546.5    78.3  4596.5    76.8  4616.5      76  4656.5    75.7  4717.3    77.1
  4737.3    76.7  4757.3    76.8  4758.8   76.74  4767.3    76.4  4800.7   77.54
  4817.3    78.1  4851.8    78.2  4858.2   77.92  4881.8    76.9 4894.09   77.07
  4894.2   77.07 4894.31   77.07  4917.4   77.38  4925.7   77.29  4928.5   77.26
  4962.3    76.7  4974.4   73.81 4978.61      72  4978.7   71.96  4978.8   71.92
  4990.4   66.93  4990.5   66.18  4990.7   64.67    4993   62.73  4998.7    62.7
  5004.9   63.22  5009.2   64.35  5009.9   67.08    5010   67.47 5021.09   71.88
  5021.2   71.93  5021.3   71.97  5028.5   74.83  5051.6   76.86  5059.1   77.52
  5079.3   77.38 5103.89    77.2    5104    77.2 5104.11    77.2  5109.1   77.17
    5120   77.09  5168.5   77.03  5187.7   77.07  5211.8   77.12    5239   77.29
  5239.9   77.28  5260.4   77.12  5302.3    76.8  5308.8    76.9  5338.8    77.4
  5358.8    77.4  5378.8    77.8
BR D #Mann= 3
  4546.5     .99  4974.4     .02  5028.5      .1
BR D Banks=4974.4,5028.5
BC Design=,, 0 ,, 0 ,,,,,,

Type RM Length L Ch R = 1 ,1258.3  ,116.7,116.7,116.7
BEGIN DESCRIPTION:
Downstream Section of Bridge/Culvert/Weir
END DESCRIPTION:
XS GIS Cut Line= 6
      3117615.69      13911494.2      3117383.64     13911620.76
      3117310.64     13911661.71      3117218.05     13911711.57
      3117129.03      13911754.3      3116870.45     13911862.68
#Sta/Elev= 30
  4546.5   78.33  4596.5   76.83  4616.5   76.03  4656.5   75.73  4717.3   77.13
  4737.3   76.73  4757.3   76.83  4767.3   76.43  4817.3   78.13  4851.8   78.23
  4881.8   76.93  4917.4   77.41  4962.3   76.73  4974.4   73.84  4990.4   66.96
  4990.7    64.7    4993   62.76  4998.7   62.73  5004.9   63.25  5009.2   64.38
    5010    67.5  5028.5   74.86  5059.1   77.55    5120   77.12  5168.5   77.06
    5239   77.32  5302.3   76.83  5338.8   77.43  5358.8   77.43  5378.8   77.83
#Mann= 3 , 1 , 0
  4546.5     .99       0  4974.4     .02       0  5028.5      .1       0
#XS Ineff= 2 , 0
       0    4968    78.7    5031       0    76.3
Permanent Ineff=
       F       F
Bank Sta=4974.4,5028.5
XS Rating Curve= 0
Exp/Cntr=.5,.3

Type RM Length L Ch R = 1 ,1141.6  ,34.2,34.2,34.2
BEGIN DESCRIPTION:
Upstream Section of Bridge/Culvert/Weir
END DESCRIPTION:
XS GIS Cut Line= 5
      3117391.34     13911533.74      3117190.79     13911626.98
      3117160.69     13911643.26      3117138.03     13911655.52
      3116906.46     13911752.47
#Sta/Elev= 22
  4760.5   76.99  4833.4   77.42  4920.9   76.21    4944   75.42  4957.3   74.96
  4979.5   73.72  4985.4   70.03    4991   66.53  4991.3   63.29  4997.1   62.38
  5000.5   62.13    5005   62.45  5008.6   63.18  5008.8   66.72  5014.9   70.48
  5020.1   73.69  5041.1   74.19  5068.9   74.59  5099.1   75.03  5163.6   75.45
  5257.5   75.83  5292.7   77.11
#Mann= 5 , 1 , 0
  4760.5      .2       0    4944     .08       0  4979.5     .02       0
  5020.1     .08       0  5068.9      .2       0
#XS Ineff= 2 , 0
       0  4984.8    70.3  5014.8       0    70.3
Permanent Ineff=
       F       F
Bank Sta=4979.5,5020.1
XS Rating Curve= 0
Exp/Cntr=.5,.3

Type RM Length L Ch R = 2 ,1124.5  ,,,
BEGIN DESCRIPTION:
CONCRETE CHECK STRUCTURE
Structure ID: P55-2
END DESCRIPTION:
Bridge Culvert--1,0,-1,-1, 0
Deck Dist Width WeirC Skew NumUp NumDn MinLoCord MaxHiCord MaxSubmerge Is_Ogee
10,14.2,3,0, 22, 22, , , .95, 0, 1,1,,
  4760.5  4833.4  4920.9    4944  4957.3  4979.5  4985.4    4991  4991.3  4997.1
  5000.5    5005  5008.6  5008.8  5014.9  5020.1  5041.1  5068.9  5099.1  5163.6
  5257.5  5292.7
   76.88   77.31    76.1   75.31   74.85   73.61   70.29    70.3    70.3   70.32
   70.33   70.34   70.35   70.35   70.38   73.58   74.08   74.48   74.92   75.34
   75.72      77
   76.88   77.31    76.1   75.31   74.85   73.61   69.92   66.42   63.18   62.27
   62.02   62.34   63.07   66.61   70.37   73.58   74.08   74.48   74.92   75.34
   75.72      77
  4760.5  4833.4  4920.9    4944  4957.3  4979.5  4985.4    4991  4991.3  4997.1
  5000.5    5005  5008.6  5008.8  5014.9  5020.1  5041.1  5068.9  5099.1  5163.6
  5257.5  5292.7
   76.88   77.31    76.1   75.31   74.85   73.61   70.29    70.3    70.3   70.32
   70.33   70.34   70.35   70.35   70.38   73.58   74.08   74.48   74.92   75.34
   75.72      77
   76.86   77.29   76.08   75.29   74.83   73.59    69.9    66.4   63.16   62.25
      62   62.32   63.05   66.59   70.35   73.56   74.06   74.46    74.9   75.32
    75.7   76.98
BR Coef= 1 , 0 , 0 ,1.25, 0 ,,,.8,-1,2,0,
WSPro=,,,, 1 ,,,, 0 ,,,, 0 ,,,,-1 ,-1 ,-1 , 0 , 0 , 0 , 0 , 0
Culvert=1,4.5,,14.2,.015,.5,1,1,3,62.08,5000,62.2,5000,Culvert #1  , 0 ,10
Culvert Bottom n=.015
BR U #Sta/Elev= 22
  4760.5   76.88  4833.4   77.31  4920.9    76.1    4944   75.31  4957.3   74.85
  4979.5   73.61  4985.4   69.92    4991   66.42  4991.3   63.18  4997.1   62.27
  5000.5   62.02    5005   62.34  5008.6   63.07  5008.8   66.61  5014.9   70.37
  5020.1   73.58  5041.1   74.08  5068.9   74.48  5099.1   74.92  5163.6   75.34
  5257.5   75.72  5292.7      77
BR U #Mann= 5
  4760.5      .2    4944     .08  4979.5     .02  5020.1     .08  5068.9      .2
BR U Banks=4979.5,5020.1
BR D #Sta/Elev= 22
  4760.5   76.86  4833.4   77.29  4920.9   76.08    4944   75.29  4957.3   74.83
  4979.5   73.59  4985.4    69.9    4991    66.4  4991.3   63.16  4997.1   62.25
  5000.5      62    5005   62.32  5008.6   63.05  5008.8   66.59  5014.9   70.35
  5020.1   73.56  5041.1   74.06  5068.9   74.46  5099.1    74.9  5163.6   75.32
  5257.5    75.7  5292.7   76.98
BR D #Mann= 5
  4760.5      .2    4944     .08  4979.5     .02  5020.1     .08  5068.9      .2
BR D Banks=4979.5,5020.1
BC Design=,, 0 ,, 0 ,,,,,,

Type RM Length L Ch R = 1 ,1107.4  ,209.3,209.3,209.3
BEGIN DESCRIPTION:
Downstream Section of Bridge/Culvert/Weir
END DESCRIPTION:
XS GIS Cut Line= 5
      3117374.93     13911503.74      3117174.39     13911596.98
      3117144.29     13911613.26      3117121.63     13911625.52
      3116890.05     13911722.46
#Sta/Elev= 22
  4760.5   76.85  4833.4   77.28  4920.9   76.07    4944   75.28  4957.3   74.82
  4979.5   73.58  4985.4   69.89    4991   66.39  4991.3   63.15  4997.1   62.24
  5000.5   61.99    5005   62.31  5008.6   63.04  5008.8   66.58  5014.9   70.34
  5020.1   73.55  5041.1   74.05  5068.9   74.45  5099.1   74.89  5163.6   75.31
  5257.5   75.69  5292.7   76.97
#Mann= 5 , 1 , 0
  4760.5      .2       0    4944     .08       0  4979.5     .02       0
  5020.1     .08       0  5068.9      .2       0
#XS Ineff= 2 , 0
       0  4984.8    70.3  5014.8       0    70.3
Permanent Ineff=
       F       F
Bank Sta=4979.5,5020.1
XS Rating Curve= 0
Exp/Cntr=.5,.3

Type RM Length L Ch R = 1 ,898.1   ,58,57.9,53.6
BEGIN DESCRIPTION:
Cross Section 898.1-Interpolated
END DESCRIPTION:
XS GIS Cut Line= 5
      3117424.85     13911413.73      3117344.86     13911417.36
      3117159.53     13911413.73      3117057.79     13911406.46
      3116866.94     13911399.76
#Sta/Elev= 25
  4694.5    76.4  4704.5    75.3  4762.4   75.55  4795.4   75.13    4831   75.34
  4875.6   75.23  4927.2    74.8  4933.4   74.75    4978   72.63  4990.8      66
  4991.2   62.38  4993.8   61.87    4999   61.66    5005   61.72  5008.8   62.35
  5009.3   65.91  5021.6   72.16  5035.6   74.94    5040   75.01  5069.1   75.44
  5116.8   75.22  5170.2   75.98    5238   74.77    5252    75.7  5252.9    76.5
#Mann= 5 , 1 , 0
  4694.5     .12       0  4927.2     .08       0    4978    .015       0
  5021.6     .08       0    5040      .1       0
#XS Ineff= 2 , 0
       0                  5170.2       0   75.98
Permanent Ineff=
       F       F
Bank Sta=4978,5021.6
XS Rating Curve= 0
Exp/Cntr=.5,.3

Type RM Length L Ch R = 1 ,840.2   ,56.4,56.4,56.4
BEGIN DESCRIPTION:
Upstream Section of Bridge/Culvert/Weir
END DESCRIPTION:
XS GIS Cut Line= 4
       3117376.9     13911355.64       3117180.7     13911342.55
      3117102.16     13911342.55      3116860.42      13911330.9
#Sta/Elev= 22
  4746.1   76.31    4760   75.81  4762.4   75.56  4795.4   75.14    4831   75.35
  4875.6   75.24  4933.4   74.76    4978   72.64  4990.8   66.01  4991.2   62.39
  4993.8   61.88    4999   61.67    5005   61.73  5008.8   62.36  5009.2   65.92
  5021.6   72.17  5035.6   74.95  5069.1   75.45  5116.8   75.23  5170.2   75.99
    5238   74.78  5263.3   76.11
#Mann= 3 , 1 , 0
  4746.1      .1       0    4978    .015       0  5021.6      .1       0
#XS Ineff= 2 , 0
       0    4965    76.4    5033       0    76.4
Permanent Ineff=
       F       F
Bank Sta=4978,5021.6
XS Rating Curve= 0
Exp/Cntr=.5,.3

Type RM Length L Ch R = 3 ,812.0   ,,,
BEGIN DESCRIPTION:
OLD GREENS ROAD
Structure ID: P55-1
END DESCRIPTION:
Bridge Culvert--1,0,-1,-1, 0
Deck Dist Width WeirC Skew NumUp NumDn MinLoCord MaxHiCord MaxSubmerge Is_Ogee
10,36.4,2.6,0, 45, 45, , , .95, 0, 1,1,,
  4746.1    4760  4761.3  4762.4  4795.4    4831  4840.8  4875.6  4900.4  4933.4
    4955 4968.99  4969.1 4969.21  4975.1 4975.21  4975.3    4978  4990.8  4990.9
  4991.2  4993.8    4999    5005  5008.8  5009.2  5009.3  5021.6 5023.79  5023.9
    5024 5029.89    5030 5030.11  5035.6  5052.4  5069.1  5116.8  5131.9  5170.2
  5187.3  5237.2    5238    5260  5263.3
    76.3   76.48    76.5    76.5    76.5    76.5    76.5   76.54   76.57   76.47
   76.41    76.4    78.9    78.9   78.89   78.89   78.89   78.89   78.87   78.87
   78.87   78.87   78.87   78.86   78.86   78.86   78.85   78.84   78.84   78.84
   78.84   78.86   78.86   76.36   76.37   76.41   76.44   76.52   76.54   76.68
   76.74   76.57   76.57   76.55    76.1
    76.3    75.8   75.66   75.55   75.13   75.34   75.32   75.23   75.02   74.75
   73.72   73.06   73.05   73.05   72.77   72.76   74.21   74.21   74.19   74.19
   74.19   74.19   74.19   74.18   74.18   74.18   74.17   74.16   74.16   72.62
   72.64   73.81   73.83   73.85   74.94   75.19   75.44   75.22   75.43   75.98
   75.67   74.78   74.77   75.93    76.1
  4746.1    4760  4761.3  4762.4  4795.4    4831  4840.8  4875.6  4900.4  4933.4
    4955 4968.99  4969.1 4969.21  4975.1 4975.21  4975.3    4978  4990.8  4990.9
  4991.2  4993.8    4999    5005  5008.8  5009.2  5009.3  5021.6 5023.79  5023.9
    5024 5029.89    5030 5030.11  5035.6  5052.4  5069.1  5116.8  5131.9  5170.2
  5187.3  5237.2    5238    5260  5263.3
    76.3   76.48    76.5    76.5    76.5    76.5    76.5   76.54   76.57   76.47
   76.41    76.4    78.9    78.9   78.89   78.89   78.89   78.89   78.87   78.87
   78.87   78.87   78.87   78.86   78.86   78.86   78.85   78.84   78.84   78.84
   78.84   78.86   78.86   76.36   76.37   76.41   76.44   76.52   76.54   76.68
   76.74   76.57   76.57   76.55    76.1
   76.12   75.62   75.48   75.37   74.95   75.16   75.14   75.05   74.84   74.57
   73.54   72.88   72.87   72.87   72.59   72.58   74.03   74.03   74.01   74.01
   74.01   74.01   74.01      74      74      74   73.99   73.98   73.98   72.44
   72.46   73.63   73.65   73.67   74.76   75.01   75.26   75.04   75.25    75.8
   75.49    74.6   74.59   75.75   75.92
Abutment Skew #Up #Dn= , 2 , 2
  4975.1  4990.9
   74.21    65.1
  4975.1  4990.9
   74.03   64.92
Abutment Skew #Up #Dn= , 2 , 2
  5009.3 5023.99
   65.96   74.16
  5009.3 5023.99
   65.78   73.98
BR Coef= 1 , 1 , 0 ,1.25, 0 ,,,.8,0,2,0,
WSPro=,,,, 1 ,,,, 0 ,,,, 0 ,,,,-1 ,-1 ,-1 , 0 , 0 , 0 , 0 , 0
BR U #Sta/Elev= 45
  4746.1    76.3    4760    75.8  4761.3   75.66  4762.4   75.55  4795.4   75.13
    4831   75.34  4840.8   75.32  4875.6   75.23  4900.4   75.02  4933.4   74.75
    4955   73.72 4968.99   73.06  4969.1   73.05 4969.21   73.05  4975.1   72.77
 4975.21   72.76  4975.3   72.76    4978   72.63  4990.8      66  4990.9    65.1
  4991.2   62.38  4993.8   61.87    4999   61.66    5005   61.72  5008.8   62.35
  5009.2   65.91  5009.3   65.96  5021.6   72.16 5023.79   72.59  5023.9   72.62
    5024   72.64 5029.89   73.81    5030   73.83 5030.11   73.85  5035.6   74.94
  5052.4   75.19  5069.1   75.44  5116.8   75.22  5131.9   75.43  5170.2   75.98
  5187.3   75.67  5237.2   74.78    5238   74.77    5260   75.93  5263.3    76.1
BR U #Mann= 3
  4746.1      .1    4978    .015  5021.6      .1
BR U Banks=4978,5021.6
BR D #Sta/Elev= 45
  4746.1   76.12    4760   75.62  4761.3   75.48  4762.4   75.37  4795.4   74.95
    4831   75.16  4840.8   75.14  4875.6   75.05  4900.4   74.84  4933.4   74.57
    4955   73.54 4968.99   72.88  4969.1   72.87 4969.21   72.87  4975.1   72.59
 4975.21   72.58  4975.3   72.58    4978   72.45  4990.8   65.82  4990.9   64.92
  4991.2    62.2  4993.8   61.69    4999   61.48    5005   61.54  5008.8   62.17
  5009.2   65.73  5009.3   65.78  5021.6   71.98 5023.79   72.41  5023.9   72.44
    5024   72.46 5029.89   73.63    5030   73.65 5030.11   73.67  5035.6   74.76
  5052.4   75.01  5069.1   75.26  5116.8   75.04  5131.9   75.25  5170.2    75.8
  5187.3   75.49  5237.2    74.6    5238   74.59    5260   75.75  5263.3   75.92
BR D #Mann= 3
  4746.1      .1    4978    .015  5021.6      .1
BR D Banks=4978,5021.6
BC Design=,, 0 ,, 0 ,,,,,,

Type RM Length L Ch R = 1 ,783.8   ,270.2,270.2,270.2
BEGIN DESCRIPTION:
Downstream Section of Bridge/Culvert/Weir
END DESCRIPTION:
XS GIS Cut Line= 4
       3117380.1     13911299.33       3117183.9     13911286.25
      3117105.36     13911286.25      3116863.61     13911274.59
#Sta/Elev= 22
  4746.1   76.12    4760   75.62  4762.4   75.37  4795.4   74.95    4831   75.16
  4875.6   75.05  4933.4   74.57    4978   72.45  4990.8   65.82  4991.2    62.2
  4993.8   61.69    4999   61.48    5005   61.54  5008.8   62.17  5009.2   65.73
  5021.6   71.98  5035.6   74.76  5069.1   75.26  5116.8   75.04  5170.2    75.8
    5238   74.59  5263.3   75.92
#Mann= 3 , 1 , 0
  4746.1      .1       0    4978    .015       0  5021.6      .1       0
#XS Ineff= 2 , 0
       0    4965    75.7    5033       0    76.2
Permanent Ineff=
       F       F
Bank Sta=4978,5021.6
XS Rating Curve= 0
Exp/Cntr=.5,.3

Type RM Length L Ch R = 1 ,513.6   ,0,0,0
BEGIN DESCRIPTION:
Cross Section 513.6
END DESCRIPTION:
XS GIS Cut Line= 2
      3117345.59     13911023.97      3116945.63     13911029.68
#Sta/Elev= 19
  4793.9    79.8  4833.9    78.9  4863.9    78.8  4903.9    76.4  4939.8    75.8
  4958.6    75.9  4975.1      75    4991    66.2  4991.2      62    5000    61.5
  5008.7      62  5009.2    66.1    5025    74.6    5030   74.22  5044.8   74.31
  5153.9    74.3  5163.9    74.5  5183.9    75.9  5193.9    76.1
#Mann= 3 , 1 , 0
  4793.9      .1       0  4975.1    .015       0    5025      .1       0
Bank Sta=4975.1,5025
XS Rating Curve= 0
Exp/Cntr=.3,.1

Chan Stop Cuts=-1
